--- Case.prj (project) ---

Proj Title=A2C-EA5
Current Plan=p01
Default Exp/Contr=0.3,0.1
SI Units
Geom File=g01
Unsteady File=u01
Plan File=p01
Y Axis Title=Elevation
X Axis Title(PF)=Main Channel Distance
X Axis Title(XS)=Station
BEGIN DESCRIPTION:
A2C-EA5
END DESCRIPTION:
DSS File=dss

--- Case.p01 (plan) ---

Plan Title=Main
Program Version=6.60
Short Identifier=main
Simulation Date=01JAN2000,0000,02JAN2000,0600
Geom File=g01
Flow File=u01
Subcritical Flow
K Sum by GR= 0
Std Step Tol= 0.01
Critical Tol= 0.01
Num of Std Step Trials= 20
Max Error Tol= 0.3
Flow Tol Ratio= 0.001
Split Flow NTrial= 30
Split Flow Tol= 0.02
Split Flow Ratio= 0.02
Log Output Level= 0
Friction Slope Method= 1
Unsteady Friction Slope Method= 2
Unsteady Bridges Friction Slope Method= 1
Parabolic Critical Depth
Global Vel Dist= 0 , 0 , 0
Global Log Level= 0
CheckData=True
Encroach Param=-1 ,0,0, 0
Computation Interval=1SEC
Output Interval=1MIN
Instantaneous Interval=1HOUR
Mapping Interval=1MIN
Computation Time Step Use Courant=        -1
Computation Time Step Use Time Series=    0
Computation Time Step Max Courant=1
Computation Time Step Min Courant=0.45
Computation Time Step Count To Double=4
Computation Time Step Max Doubling=3
Computation Time Step Max Halving=6
Computation Time Step Residence Courant=0
Run HTab=-1
Run UNet=-1
Run Sediment= 0
Run PostProcess= 0
Run WQNet= 0
Run RASMapper= 0
UNET Theta= 1
UNET Theta Warmup= 1
UNET ZTol= 0.02
UNET ZSATol= 0.02
UNET MxIter= 20
UNET Max Iter WO Improvement= 0
UNET MaxInSteps= 0
UNET DtIC= 0
UNET DtMin= 0
UNET MaxCRTS= 20
UNET WFStab= 2
UNET SFStab= 1
UNET WFX= 1
UNET SFX= 1
UNET Gravity=9.81
UNET 1D Methodology=Finite Difference
UNET DSS MLevel= 4
UNET Pardiso=0
UNET DZMax Abort= 100
UNET Use Existing IB Tables=-1
UNET Froude Reduction=False
UNET Froude Limit= 1
UNET Froude Power= 10
UNET D1 Cores= 0
UNET D2 Coriolis=0
UNET D2 Theta= 1
UNET D2 Theta Warmup= 1
UNET D2 Z Tol= 0.01
UNET D2 Volume Tol= 0.01
UNET D2 Max Iterations= 20
UNET D2 Equation= 1
UNET D2 RampUpFraction=0.1
UNET D2 TimeSlices= 1
UNET D2 Turbulence Formulation=None
UNET D2 BCVolumeCheck=0
UNET D2 Cores=0
UNET D2 SolverType=Pardiso (Direct)
UNET D2 Name=Strip
UNET D2 Coriolis=0
UNET D2 Theta= 1
UNET D2 Theta Warmup= 1
UNET D2 Z Tol= 0.01
UNET D2 Volume Tol= 0.01
UNET D2 Max Iterations= 20
UNET D2 Equation= 1
UNET D2 RampUpFraction=0.1
UNET D2 TimeSlices= 1
UNET D2 Turbulence Formulation=None
UNET D2 BCVolumeCheck=0
UNET D2 Cores=0
UNET D2 SolverType=Pardiso (Direct)
UNET D1D2 MaxIter= 0
UNET D1D2 ZTol=0.02
UNET D1D2 QTol=1
DSS File=dss
Write IC File= 0
Write IC File at Fixed DateTime=0
Write IC File at Sim End=0
Echo Input=False
Echo Parameters=False
Echo Output=False
Write Detailed= 0
HDF Write Warmup=0
HDF Write Time Slices=0
HDF Flush=0
HDF Additional Output Variable=Cell Velocity
HDF Additional Output Variable=Face Flow
HDF Compression= 1
HDF Chunk Size= 1
HDF Spatial Parts= 1
HDF Use Max Rows=0
HDF Fixed Rows= 1

--- Case.u01 (unsteady flow) ---

Flow Title=main
Program Version=6.60
Use Restart= 0
Boundary Location=                ,                ,        ,        ,                ,Strip           ,                ,Inflow
Interval=1MIN
Flow Hydrograph= 1802
  0.0000  0.0000  0.0000  0.0000  0.0000  0.0000600.00001200.0001800.0002400.000
3000.0003000.0003000.0003000.0003000.0003000.0003000.0003000.0003000.0003000.000
3000.0002962.5002925.0002887.5002850.0002812.5002775.0002737.5002700.0002662.500
2625.0002587.5002550.0002512.5002475.0002437.5002400.0002362.5002325.0002287.500
2250.0002212.5002175.0002137.5002100.0002062.5002025.0001987.5001950.0001912.500
1875.0001837.5001800.0001762.5001725.0001687.5001650.0001612.5001575.0001537.500
1500.0001462.5001425.0001387.5001350.0001312.5001275.0001237.5001200.0001162.500
1125.0001087.5001050.0001012.500975.0000937.5000900.0000862.5000825.0000787.5000
750.0000712.5000675.0000637.5000600.0000562.5000525.0000487.5000450.0000412.5000
375.0000337.5000300.0000262.5000225.0000187.5000150.0000112.5000 75.0000 37.5000
  0.0000  0.0000  0.0000  0.0000  0.0000  0.0000  0.0000  0.0000  0.0000  0.0000
  0.0000  0.0000  0.0000  0.0000  0.0000  0.0000  0.0000  0.0000  0.0000  0.0000
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Stage Hydrograph TW Check=0
Flow Hydrograph Slope= 0.001
Use DSS=False
Use Fixed Start Time=False
Is Critical Boundary=False
Precipitation Mode=Disable
Wind Mode=No Wind Forces
Met BC=Precipitation|Mode=None
Met BC=Evapotranspiration|Mode=None

--- Case.g01 (geometry) ---

Geom Title=A2C-EA5
Program Version=6.60

Storage Area=Strip           ,738698.4609375,4835612.8125
Storage Area Surface Line= 6
   732324.843750  4830731.750000
   738761.875000  4837105.375000
   737731.312500  4840688.375000
   745024.515625  4840583.000000
   740759.578125  4839742.687500
   732324.843750  4830731.750000
Storage Area Type= 0
Storage Area Is2D=-1
Storage Area Point Generation Data=,,50,50
Storage Area 2D Points= 7643
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Storage Area Mannings=0.04
2D Cell Volume Filter Tolerance=0.003
2D Cell Minimum Area Fraction=0.01
2D Face Profile Filter Tolerance=0.003
2D Face Area Elevation Profile Filter Tolerance=0.003
2D Face Area Elevation Conveyance Ratio=0.02
2D Face Area Laminar Depth=0.2

BC Line Name=Inflow
BC Line Storage Area=Strip
BC Line Start Position= 732595.0 , 4830480.0
BC Line Middle Position= 732690.0 , 4830385.0
BC Line End Position= 732785.0 , 4830290.0
BC Line Arc= 2
   732595.000000  4830480.000000   732785.000000  4830290.000000
LCMann Table=0

Chan Stop Cuts=-1
